HEC-RAS study HNSCK.prj: HNSCK

--- HNSCK.g01 (geometry) --- (continued)

Type RM Length L Ch R = 1 ,59445   ,61.2,61.4,65.3
XS GIS Cut Line= 6
     2065162.005      173583.992     2065500.544      174148.995
     2065563.478       174216.27     2065691.516      174211.929
     2066038.799      174439.702     2066184.138      174613.405
#Sta/Elev= 30
       0  1941.8    28.9 1941.15   60.89 1937.12   63.57 1936.28  110.211928.711
   166.1 1926.81   192.3 1929.83  206.211935.722  228.321940.732  237.531941.415
  283.841941.894     343 1940.89   431.4 1928.53  481.741924.815  505.891923.198
  551.521920.291   561.41919.896   689.2 1917.13   705.1 1912.78   711.4 1911.87
   724.1  1912.8  736.391915.126  765.06 1915.66 1072.381915.778 1234.351917.561
  1292.9 1918.68  1393.2  1924.9 1479.831934.812 1490.011937.193  1522.6 1940.52
#Mann= 20 ,-1 , 0
       0     .08       0   60.89     .06       0   63.57     .08       0
  110.21     .06       0  206.21     .12       0  228.32    .016       0
  237.53     .06       0  283.84    .016       0  481.74     .06       0
  505.89    .016       0  551.52     .08       0   561.4    .016       0
   705.1    .045       0   724.1     .12       0  736.39    .016       0
  765.06     .06       0 1072.38    .016       0 1234.35     .06       0
 1479.83     .08       0 1490.01    .016       0
Bank Sta=705.1,724.1
XS Rating Curve= 0 ,0
Exp/Cntr=0.3,0.1

Type RM Length L Ch R = 1 ,59383.6 ,245.5,237.3,223.8
XS GIS Cut Line= 6
     2065073.698      173684.286     2065433.143      174165.829
     2065528.756      174266.183     2065656.794      174261.843
     2065995.336      174483.197     2066132.055      174663.318
#Sta/Elev= 30
       0    1970    39.2 1949.09      98 1929.82   127.4 1929.31   140.4 1932.66
  150.761938.542   169.8 1949.12  180.951950.702   241.7 1951.36  280.111954.121
   329.8 1959.02   382.1 1958.71   431.1 1952.11  466.241943.571  526.591928.022
  538.381926.027  569.611921.177  654.11 1917.33   668.6 1917.12   676.8 1912.58
   681.5    1912   697.6 1912.43   713.7 1914.93 1270.411916.687 1279.731917.451
 1294.691918.833    13301921.283 1370.611923.453  1410.81926.232  1498.2 1933.37
#Mann= 17 ,-1 , 0
       0     .06       0  150.76     .12       0  180.95     .08       0
  280.11     .06       0  466.24     .12       0  526.59     .08       0
  538.38     .12       0  569.61     .06       0  654.11     .12       0
   676.8    .045       0   697.6     .06       0 1270.41    .016       0
 1279.73     .06       0 1294.69     .08       0    1330     .06       0
 1370.61    .016       0  1410.8     .06       0
Bank Sta=676.8,697.6
XS Rating Curve= 0 ,0
Exp/Cntr=0.3,0.1

Type RM Length L Ch R = 1 ,59146.3 ,502.9,500.5,492.6
XS GIS Cut Line= 3
     2065222.766      174410.497     2065409.398      174412.667
     2066084.312      174707.806
#Sta/Elev= 30
       0 2028.84    16.4 2021.14    39.3 2007.53    65.5 1989.98    88.4 1973.21
    98.2 1966.95   114.6 1954.67   137.5 1939.78   157.2 1930.15   176.8 1922.47
  191.911921.055     203  1917.6   209.6 1916.69   248.8 1914.76   281.6 1914.38
   293.1 1912.71   301.2 1910.56   304.5 1910.34   314.3 1912.44   320.9 1914.18
     334 1914.54   356.9 1914.01   468.2 1914.72   510.8 1914.17   651.5 1914.93
   743.2 1917.99   851.2 1923.46   903.6 1927.31  915.191928.974   923.3 1930.09
#Mann= 5 ,-1 , 0
       0     .12       0  191.91     .06       0   293.1    .045       0
   314.3     .06       0  915.19     .08       0
Bank Sta=293.1,314.3
XS Rating Curve= 0 ,0
Exp/Cntr=0.3,0.1

Type RM Length L Ch R = 1 ,58645.8 ,527.2,535.3,528.5
XS GIS Cut Line= 2
     2065133.791      174814.143     2066036.569      175009.455
#Sta/Elev= 30
       0 2026.88    16.4 2018.84    26.2 2012.59    39.3 2002.98    65.5 1985.72
   104.8 1956.91   140.8 1932.69   150.7 1926.74  167.761919.374   186.7 1914.96
   203.1 1912.99   242.4 1912.13  266.111912.497  283.931912.417   288.2 1911.12
   298.1 1909.37   307.9 1910.35   317.7 1912.23   330.8 1912.55   412.7 1911.92
   442.2 1912.65   507.7 1912.08   533.9    1913   563.4 1912.53   694.4 1913.03
   720.6 1914.23   763.2    1920   841.8 1922.96   897.5 1926.21   923.7  1928.7
#Mann= 6 ,-1 , 0
       0     .12       0  167.76     .06       0  266.11     .12       0
  283.93     .06       0   288.2    .045       0   307.9     .06       0
Bank Sta=288.2,307.9
XS Rating Curve= 0 ,0
Exp/Cntr=0.3,0.1

Type RM Length L Ch R = 1 ,58110.4 ,218.4,221.7,224.6
XS GIS Cut Line= 3
     2065112.089      175159.195     2065205.405       175243.83
     2066040.909      175436.973
#Sta/Elev= 30
       0 1999.61    32.3 1981.24    67.8 1959.36   109.8 1931.81  127.141921.428
   132.5 1918.08   145.6  1912.7     162 1910.11   188.2 1909.76   194.7 1907.98
   207.8 1907.11   214.9 1907.94   224.2 1909.84   276.5 1910.38   351.8 1910.63
     378 1909.89   417.3 1911.37   525.3  1910.7   672.6 1911.82   695.5  1913.7
   728.2  1918.9   780.6 1922.79     810 1925.69  825.021927.972   839.5 1931.14
  859.751931.596   875.5 1937.06  888.071939.327   918.1 1943.95   983.5 1949.55
#Mann= 7 ,-1 , 0
       0     .12       0  127.14     .06       0   194.7    .045       0
   214.9     .06       0  825.02    .016       0  859.75     .12       0
  888.07     .06       0
Bank Sta=194.7,214.9
XS Rating Curve= 0 ,0
Exp/Cntr=0.3,0.1

Type RM Length L Ch R = 1 ,57888.8 ,347.4,345.8,298.8
XS GIS Cut Line= 3
     2065036.135      175289.403      2065114.26      175417.442
     2065928.062      175588.883
#Sta/Elev= 30
       0 2003.68    26.1 1994.35    42.4 1987.04    91.3 1961.56   110.9 1950.52
     150 1924.08   163.1 1917.49   172.9 1913.52  185.421912.062   225.3 1909.23
     258 1909.52   280.1 1907.96   290.8  1906.3   297.3 1907.51   307.2 1909.66
   372.6 1908.79   451.2 1910.03   605.1 1909.61   677.2 1911.54  724.421914.532
     759 1917.37   778.6 1917.28   788.5 1919.55   801.6 1924.66   814.7 1923.48
  853.361925.121   873.6  1929.2   893.2 1928.92  899.371930.393   981.7  1936.8
#Mann= 7 ,-1 , 0
       0     .12       0  185.42     .06       0   280.1    .045       0
   297.3     .06       0  724.42     .12       0  853.36    .016       0
  899.37     .06       0
Bank Sta=280.1,297.3
XS Rating Curve= 0 ,0
Exp/Cntr=0.3,0.1

Type RM Length L Ch R = 1 ,57543   ,65.1,63,68.4
XS GIS Cut Line= 4
      2064968.86      175612.754      2065120.77      175682.199
     2065207.575       175701.73      2065897.68      175630.115
#Sta/Elev= 30
       0 1914.23      36 1914.51   90.721913.622   144.1 1912.71   189.3 1910.28
  259.82 1908.47   265.8 1906.51   269.1 1905.44   278.9 1905.05   285.5 1905.36
   288.7  1906.3  289.521906.663     292 1907.76   298.6 1908.62   373.8 1907.85
  645.891909.445   684.7 1909.47   714.2 1910.61   730.6  1912.7   756.7 1917.87
  794.381922.843  808.431924.019   835.3 1925.68   845.1 1927.42  869.791926.876
   874.5 1927.53   881.1 1930.76   884.4 1931.39     904 1931.95   949.8 1935.52
#Mann= 10 ,-1 , 0
       0     .06       0   90.72    .016       0  259.82     .12       0
   265.8    .045       0   288.7     .12       0  289.52     .06       0
  645.89     .12       0  794.38     .06       0  808.43    .016       0
  869.79     .06       0
Bank Sta=265.8,288.7
XS Rating Curve= 0 ,0
Exp/Cntr=0.3,0.1

Type RM Length L Ch R = 1 ,57480   ,426.7,430.6,422.9
XS GIS Cut Line= 4
      2064962.35      175664.837      2065114.26      175734.282
     2065201.065      175753.813     2065891.169      175682.199
#Sta/Elev= 30
       0 1917.46   13.971916.092   48.861914.599    78.6 1913.48  272.821909.738
   288.7 1908.77   310.9 1906.06   321.5 1904.63   334.6 1904.72   341.1 1906.32
   347.6 1907.56   357.5  1907.9   413.1 1907.73     436 1908.41   511.3 1908.82
   576.7 1907.96  625.721909.229   717.5 1908.93   750.2 1909.62     760 1910.48
   773.1 1912.64   802.5 1919.86   817.51922.721     832 1924.54   838.5 1925.97
   864.7 1924.61  871.981928.778   874.5 1930.18   877.8 1930.97   949.8 1940.51
#Mann= 9 ,-1 , 0
       0     .08       0   13.97    .016       0   48.86     .06       0
  272.82     .12       0   310.9    .045       0   341.1     .06       0
  625.72     .12       0   817.5    .016       0  871.98     .06       0
Bank Sta=310.9,341.1
XS Rating Curve= 0 ,0
Exp/Cntr=0.3,0.1

Type RM Length L Ch R = 1 ,57049.4 ,736,749.2,758.2
XS GIS Cut Line= 3
     2064979.711      176035.931     2065821.725      175946.955
     2066095.162      175951.296
#Sta/Elev= 30
       0 1968.56    55.6 1935.59   101.3 1917.96   124.2  1911.6   166.7 1909.67
   225.6 1908.65     340 1909.43   379.2 1907.01  411.151906.758   431.5 1906.45
  440.86 1904.86   446.3 1903.68   454.4 1903.12   461.3  1903.8   470.8 1905.58
   523.1 1907.23   735.6 1907.36   751.9 1908.82   797.3 1916.21   817.3 1920.01
  827.011924.657   843.4 1925.65  848.43 1929.52   853.2  1932.7   866.2 1935.16
   892.3 1942.92   931.4 1949.66   963.9 1953.39  1055.1 1960.98  1120.2 1968.78
#Mann= 8 ,-1 , 0
       0     .06       0  411.15     .12       0  440.86     .06       0
   446.3    .045       0   461.3     .06       0   797.3     .08       0
  827.01    .016       0  848.43     .06       0
Bank Sta=446.3,461.3
XS Rating Curve= 0 ,0
Exp/Cntr=0.3,0.1

Type RM Length L Ch R = 1 ,56300.2 ,462.6,466.7,468.9
XS GIS Cut Line= 3
     2064994.902      176239.924     2065090.388      176255.115
     2065919.381      176571.955
#Sta/Elev= 30
       0 1983.53    25.8 1964.96    54.8 1942.67    70.9 1932.53    90.2 1921.16
   106.5 1914.12  116.061910.994   122.9 1908.27   129.4  1904.1   132.7 1902.08
   139.3 1901.19   152.4 1903.12   211.3 1904.47   293.2 1903.88     375 1905.35
   551.9 1905.24  658.831907.913  666.361908.028   686.2 1908.21  710.351910.401
   738.6 1913.88   807.3 1917.95     827 1921.15   836.8 1925.05  841.321925.843
   856.4 1925.68  863.451930.403   892.5 1941.09   928.5  1950.4   984.2 1960.32
#Mann= 9 ,-1 , 0
       0     .12       0  116.06     .06       0   129.4    .045       0
   152.4     .06       0  658.83     .12       0  666.36     .06       0
  710.35     .12       0  841.32    .016       0  863.45     .06       0
#XS Ineff= 2 , 0
                          490.11         1919.76
Permanent Ineff=
       F       F
Bank Sta=129.4,152.4
XS Rating Curve= 0 ,0
Exp/Cntr=0.3,0.1

Type RM Length L Ch R = 1 ,55833.5 ,899.9,900.3,894
XS GIS Cut Line= 2
     2064840.822      176632.719      2065585.18      177008.153
#Sta/Elev= 30
       0    1979     6.5 1974.91     9.8 1972.32    19.6  1964.6    42.5 1945.37
    65.4 1927.67    78.5 1916.09      85 1909.27    88.3 1906.37    94.8 1902.42
    98.1 1901.38   109.6 1899.44   117.7 1899.04   127.5 1899.65     134 1901.67
   140.6 1902.16   163.5 1902.18   179.8 1903.65     206  1903.8   241.9  1904.9
   313.9 1903.93   405.4 1905.53     461 1905.46   519.8 1904.64   666.9 1905.29
   693.1 1905.88     716 1908.15  821.491925.969   830.4 1929.64   833.7 1930.12
#Mann= 4 ,-1 , 0
       0     .12       0   109.6    .045       0   127.5     .06       0
  821.49    .016       0
#XS Ineff= 2 , 0
                          375.35         1918.57
Permanent Ineff=
       F       F
Bank Sta=109.6,127.5
XS Rating Curve= 0 ,0
Exp/Cntr=0.3,0.1

Type RM Length L Ch R = 1 ,54933.2 ,193.6,194.1,193.7
XS GIS Cut Line= 4
      2064497.94      177086.278      2064964.52      177364.056
      2065122.94      177405.289     2065450.631      177624.473
#Sta/Elev= 30
       0 1930.04    19.6 1917.47      36 1909.37    45.8 1906.34   63.911905.192
  325.671902.886  371.591902.188  417.661902.333  429.341902.428  486.411901.931
  490.961901.684  509.611901.344  554.311900.517  584.321899.424  614.851897.806
   617.3 1897.41   624.9 1896.84   632.3 1897.74   641.2 1900.34  681.421901.152
   741.91901.488  793.641907.577   872.9 1916.07  884.051919.839   905.4 1919.93
  914.551923.462   931.5 1927.57   977.1  1944.8  1019.5 1958.34  1100.9  1975.9
#Mann= 19 ,-1 , 0
       0     .12       0   63.91     .06       0  325.67    .016       0
  371.59     .12       0  417.66     .06       0  429.34     .12       0
  486.41    .016       0  490.96     .06       0  509.61    .016       0
  554.31     .06       0  584.32     .12       0  614.85     .06       0
   617.3    .045       0   632.3     .06       0  681.42    .016       0
   741.9     .12       0  793.64     .06       0  884.05    .016       0
  914.55     .12       0
Bank Sta=617.3,632.3
XS Rating Curve= 0 ,0
Exp/Cntr=0.3,0.1

Type RM Length L Ch R = 1 ,54739.1 ,433.4,444.2,451.4
XS GIS Cut Line= 4
     2064382.923      177170.914     2064988.391      177546.348
     2065146.812       177587.58     2065474.503      177806.765
#Sta/Elev= 30
       0  1934.8     6.5 1931.58    22.9 1928.46      36 1921.62   52.99 1916.24
    94.8 1907.21   127.4 1904.19  403.131901.906  446.911902.235   650.3 1902.02
  720.741899.421  736.281899.414   771.4 1899.53   784.1 1897.48   794.3 1896.24
   804.1 1897.67  858.471909.616  923.221920.134   934.8 1923.27   954.3 1923.19
   965.11925.872   973.9 1926.83   983.6 1932.12  1029.2 1947.71  1071.6 1958.86
    1127 1967.16  1169.4 1964.46  1211.7 1980.26  1256.81990.446  1270.4 1992.36
#Mann= 12 ,-1 , 0
       0     .12       0   52.99     .06       0  403.13     .12       0
  446.91     .06       0  720.74     .12       0  736.28     .06       0
   784.1    .045       0   804.1     .06       0  858.47     .12       0
  923.22    .016       0   965.1     .12       0  1256.8     .06       0
#XS Ineff= 2 , 0
           331.6 1916.71
Permanent Ineff=
       F       F
Bank Sta=784.1,804.1
XS Rating Curve= 0 ,0
Exp/Cntr=0.3,0.1

Type RM Length L Ch R = 1 ,54295   ,715,708.1,700.3
XS GIS Cut Line= 2
     2064285.266      177403.119     2065157.662      178036.799
#Sta/Elev= 30
       0 1911.17   22.151904.635      36 1902.84    91.8 1901.38   190.1 1900.74
   396.6 1900.87   471.9 1899.62   655.5  1900.3   701.4 1897.93   753.8 1899.75
     780 1899.14  807.281896.327   809.5 1895.97   819.3 1894.75   829.2 1895.85
     839 1899.04   845.6 1904.66     854 1913.73   858.7 1918.66     862 1921.09
   865.2 1922.03   884.9 1922.14   888.2 1923.85  896.071933.113   901.3 1937.38
   914.4 1943.69   960.3 1963.54   989.8 1975.24  1035.6 1991.92  1078.2 2003.96
#Mann= 7 ,-1 , 0
       0     .12       0   22.15     .06       0  807.28     .12       0
   809.5    .045       0   829.2     .12       0     854    .016       0
  896.07     .12       0
#XS Ineff= 2 , 0
          315.43 1918.83
Permanent Ineff=
       F       F
Bank Sta=809.5,829.2
XS Rating Curve= 0 ,0
Exp/Cntr=0.3,0.1

Type RM Length L Ch R = 1 ,53586.8 ,445.3,440,433.1
XS GIS Cut Line= 4
     2064016.495      178196.579     2064164.932      178201.788
     2064828.995      178402.308     2064955.839      178453.466
#Sta/Elev= 30
       0 1946.11    48.4  1928.3    80.7 1919.86   106.6  1915.2   187.8 1905.38
   220.5 1900.56   272.9 1897.28   328.5 1897.04   364.5 1894.98   420.1 1895.26
   429.9 1891.65   433.2 1891.52   446.6  1891.9   469.2 1895.41   505.2 1895.94
   528.1  1895.3   564.1 1896.38   626.2 1895.57   691.7 1897.49  778.631897.981
   793.1  1898.7  809.481901.897   825.8 1901.75  829.711904.094   835.7 1908.67
     852 1916.25   884.5 1932.82   913.8 1946.47   952.9 1962.63     979 1971.81
#Mann= 6 ,-1 , 0
       0     .06       0   429.9    .045       0   446.6     .06       0
  778.63     .12       0  809.48    .016       0  829.71     .12       0
Bank Sta=429.9,446.6
XS Rating Curve= 0 ,0
Exp/Cntr=0.3,0.1

Type RM Length L Ch R = 1 ,53146.9 ,65.1,64.4,63.5
XS GIS Cut Line= 3
     2063833.012      178663.193     2064699.763      178687.841
      2064814.78      178770.306
#Sta/Elev= 30
       0 1911.93   27.291910.559   111.2 1906.41  148.621906.891   173.4  1904.2
   206.1 1904.74   238.9 1902.57   268.3 1902.38   333.8 1899.64   428.6 1897.42
     481 1894.91  663.471893.104   726.4 1893.68   736.2  1893.1     741 1891.44
     746 1890.56   759.1  1890.9   762.4 1892.02   768.9 1893.78  799.371893.271
   824.6 1894.46   837.6 1898.83   840.9 1899.26   860.6 1899.27  867.53 1904.04
   873.5 1908.99   931.4 1940.68     954 1954.66   973.2 1964.02  1008.6 1978.55
#Mann= 8 ,-1 , 0
       0     .06       0   27.29     .12       0  148.62     .06       0
  663.47     .12       0     741    .045       0   762.4     .06       0
  799.37    .016       0  867.53     .12       0
#XS Ineff= 2 , 0
           476.2 1904.88
Permanent Ineff=
       F       F
Bank Sta=741,762.4
XS Rating Curve= 0 ,0
Exp/Cntr=0.3,0.1

Type RM Length L Ch R = 1 ,53082.5 ,218.2,218.3,216.7
XS GIS Cut Line= 3
     2063802.236      178752.103     2064686.742      178746.435
     2064786.569      178805.028
#Sta/Elev= 30
       0 1920.67    42.6 1923.17    81.9 1918.98   108.1 1919.96   114.7 1918.88
   147.4  1908.9  168.33 1906.31   199.8 1903.36  243.391902.342   298.1 1901.86
   520.9 1894.37   697.8 1893.86   710.9 1892.82   750.2  1893.2   770.1 1891.46
   776.4 1889.99   785.1 1891.41   799.4 1893.18   818.21893.065   825.6 1893.73
   838.7 1900.04   841.9 1900.53   861.6 1899.68   864.9 1901.09  871.731906.678
   881.2  1916.7   929.5  1943.5   948.8  1955.7   971.3  1966.5  1000.3 1978.27
#Mann= 7 ,-1 , 0
       0    .016       0  168.33     .12       0  243.39     .06       0
   770.1    .045       0   785.1     .06       0   818.2    .016       0
  871.73     .12       0
Bank Sta=770.1,785.1
XS Rating Curve= 0 ,0
Exp/Cntr=0.3,0.1

Type RM Length L Ch R = 1 ,52864.2 ,443.8,446.8,448.9
XS GIS Cut Line= 3
     2063849.069       178987.32      2064656.36      178948.258
     2064797.419      178876.643
#Sta/Elev= 30
       0 1938.66   30.771931.805    45.8 1926.23   70.051914.498    91.6 1903.47
   101.4 1900.48   111.3 1898.86  131.971898.104   284.7 1897.48  670.591892.346
   706.8 1893.26   723.2 1892.54     737 1890.11   746.1 1889.36     752 1890.31
   755.9 1892.03   765.7 1893.52  781.751897.986  826.551896.463   834.1 1896.73
   840.5 1898.78     847 1903.21   853.4 1909.34   856.7 1915.46   859.9 1923.96
   863.1 1930.21   872.8 1947.09     876  1950.9   895.4 1960.77   966.4  1986.3
#Mann= 9 ,-1 , 0
       0     .12       0   30.77     .06       0   70.05     .12       0
  131.97     .06       0  670.59     .12       0     737    .045       0
     752     .12       0  781.75    .016       0  826.55     .12       0
Bank Sta=737,752
XS Rating Curve= 0 ,0
Exp/Cntr=0.3,0.1

Type RM Length L Ch R = 1 ,52417.4 ,349,350,351.4
XS GIS Cut Line= 4
     2063775.284      179473.431     2063944.555      179349.733
     2064697.593      179356.244     2064845.162       178987.32
#Sta/Elev= 30
       0 1961.97    39.3 1955.12    75.3  1951.3      95 1947.86  153.421931.031
     190 1918.23  197.341916.788   206.4 1916.41     226  1910.1     262 1902.51
   291.5 1899.18   448.7 1893.59   579.6 1891.96   661.5 1893.07   828.5 1891.32
   857.9    1892   874.3 1888.97   880.9 1887.46   890.3 1888.61   913.6 1891.34
   952.9 1891.82  1135.3 1892.68  1161.4 1891.26 1230.321892.142 1232.091892.147
  1252.6 1892.02  1272.1  1895.3 1291.961896.061    1308 1901.17  1360.1 1928.22
#Mann= 8 ,-1 , 0
       0     .06       0  153.42     .12       0  197.34     .06       0
   874.3    .045       0   890.3     .06       0 1230.32     .12       0
 1232.09    .016       0 1291.96     .12       0
Bank Sta=874.3,890.3
XS Rating Curve= 0 ,0
Exp/Cntr=0.3,0.1

Type RM Length L Ch R = 1 ,52067.4 ,1002,1030.9,1055
XS GIS Cut Line= 4
     2063901.152      179703.466      2064968.86      179696.955
     2065090.388      179831.504     2065142.471      179894.438
#Sta/Elev= 30
       0 1966.93    49.1 1950.08    78.6 1938.04   90.931931.707   114.6 1918.94
  142.791905.201   150.7    1901   170.3 1895.55   229.3 1890.88   340.6 1891.03
   527.3 1889.35   563.3 1890.62   704.2 1890.58   733.6 1890.09  748.34 1887.81
   756.6 1886.21   769.7 1887.46   815.5 1890.24  896.471890.527    1035  1894.2
  1057.9 1897.66 1069.911903.265 1076.641906.108  1100.1 1906.94 1105.461908.336
  1116.3 1917.82  1119.5 1919.67  1151.9 1928.08  1288.2 1946.15  1330.7 1950.83
#Mann= 9 ,-1 , 0
       0     .06       0   90.93     .12       0  142.79     .06       0
  748.34    .045       0   769.7     .06       0  896.47     .12       0
 1069.91     .08       0 1076.64    .016       0 1105.46     .06       0
#XS Ineff= 2 , 0
          325.27 1904.64
Permanent Ineff=
       F       F
Bank Sta=748.34,769.7
XS Rating Curve= 0 ,0
Exp/Cntr=0.3,0.1

Type RM Length L Ch R = 1 ,51036.5 ,846.1,843.1,838.6
XS GIS Cut Line= 3
     2063842.558      179885.758     2064142.037      179898.778
     2064448.027      180656.157
#Sta/Elev= 30
       0 1988.42    7.181986.442    39.1 1974.43   156.4 1923.98  191.521914.651
   224.8  1909.9  257.95 1903.87   299.8 1896.82   355.5 1889.86  378.751888.499
   411.3  1887.9   427.7 1884.71   437.5  1883.8   447.4 1884.74   457.2 1885.96
   496.6  1886.5   522.8 1888.19   591.7 1885.03   608.1 1887.82   719.7 1890.82
     759 1892.75   827.9 1897.58  876.311903.793     887 1905.78   903.4 1905.51
  909.541909.128   998.5 1925.75  1034.6 1928.62    1074 1929.66  1116.6 1943.25
#Mann= 9 ,-1 , 0
       0     .06       0    7.18     .12       0  191.52     .06       0
  257.95     .12       0  378.75     .06       0   427.7    .045       0
   447.4     .06       0  876.31    .016       0  909.54     .06       0
Bank Sta=427.7,447.4
XS Rating Curve= 0 ,0
Exp/Cntr=0.3,0.1

Type RM Length L Ch R = 1 ,50193.4 ,1077,1075.1,1072.2
XS GIS Cut Line= 3
     2063323.895      180109.282     2063599.503      180565.011
     2063549.589      180762.494
#Sta/Elev= 30
       0 1975.51    29.4 1965.72    52.3 1955.44    75.2 1944.12   124.2 1912.04
   143.8 1897.63   160.1 1884.27   163.4 1882.71   178.3  1881.3   192.8 1880.91
   199.3  1881.3   212.4 1884.63   235.2    1884   261.4  1885.1   277.7 1887.03
   289.41886.679   326.7 1886.73   369.2 1890.35   424.8 1893.72   480.3 1896.08
  521.031896.614   548.8 1897.22   561.7 1896.52   564.9 1896.84   568.7 1898.44
   574.6  1900.3   581.1 1901.28   639.3 1908.02   730.21914.839   736.3 1915.25
#Mann= 7 ,-1 , 0
       0     .12       0   178.3    .045       0   199.3     .12       0
   289.4     .06       0  521.03    .016       0   568.7     .06       0
   730.2     .12       0
Bank Sta=178.3,199.3
XS Rating Curve= 0 ,0
Exp/Cntr=0.3,0.1

Type RM Length L Ch R = 1 ,49118.4 ,703.3,707.3,705.7
XS GIS Cut Line= 2
     2062766.169      180604.074     2063221.898      181233.414
#Sta/Elev= 30
       0 1946.42    19.7 1935.56    45.9 1917.04    72.1 1900.81    85.2 1891.57
    88.5 1889.76    95.1 1888.55   104.9 1883.72     141 1882.14  190.311882.524
     259  1882.2  306.191880.706     318 1881.08   324.6 1877.42     341 1876.26
   347.5 1876.48   360.6 1879.01   380.3 1879.95   426.2 1879.32   488.5 1881.79
     518 1880.88     636 1884.32   652.4  1887.5   668.61893.847   681.9 1903.42
   701.6 1904.02   704.9 1905.25  712.091912.529   724.6 1919.78     777 1943.81
#Mann= 7 ,-1 , 0
       0     .12       0  190.31     .06       0  306.19     .12       0
   324.6    .045       0   347.5     .12       0   668.6    .016       0
  712.09     .12       0
#XS Ineff= 2 , 0
                          558.06         1895.05
Permanent Ineff=
       F       F
Bank Sta=324.6,347.5
XS Rating Curve= 0 ,0
Exp/Cntr=0.3,0.1

Type RM Length L Ch R = 1 ,48411.1 ,422.7,401,379.1
XS GIS Cut Line= 2
     2062206.599      180670.538     2062542.536      181157.517
#Sta/Elev= 30
       0 2005.28    22.9 1999.69      36 1994.28    45.8 1989.14    62.1 1978.72
    68.6 1973.01    88.2 1957.95   104.6 1946.48     134 1927.73   156.9 1916.53
   173.2 1907.56   196.1  1897.7   215.7 1888.28   222.3 1886.77   225.5 1885.37
   238.6 1877.51   248.4 1874.48   256.4 1873.98   264.8 1873.86   271.4 1873.98
   281.1 1874.77   294.2 1878.78   313.8 1878.61   330.1 1880.32   346.5 1883.59
   359.5 1884.13   441.3 1891.58     536 1897.22   549.1 1896.69   591.6 1898.38
#Mann= 3 ,-1 , 0
       0     .12       0   256.4    .045       0   271.4     .12       0
Bank Sta=256.4,271.4
XS Rating Curve= 0 ,0
Exp/Cntr=0.3,0.1

Type RM Length L Ch R = 1 ,48010.1 ,430.3,416.7,401.4
XS GIS Cut Line= 4
     2061800.895      181160.586     2061974.828      181102.829
     2062391.495      181102.829     2062498.812      181189.232
#Sta/Elev= 30
       0 1962.07    16.4 1962.31    32.7 1959.32    58.9 1951.85    88.4 1941.39
   147.3 1911.98   166.9 1901.84   176.7  1895.9   189.8 1891.03   199.6    1885
   212.6 1874.21   219.1 1873.23   222.3 1873.25   249.7 1873.32   261.4 1873.46
   274.4 1876.86   284.2 1876.92     294  1875.7   300.5 1877.28   313.5 1877.84
   388.4  1876.3   407.9 1877.15   420.9 1878.47   433.9  1881.8   476.2 1895.44
   492.5 1896.97   567.4 1899.08   616.3 1898.31  726.941903.857   737.7    1904
#Mann= 4 ,-1 , 0
       0     .12       0   222.3    .045       0   249.7     .12       0
  726.94     .06       0
Bank Sta=222.3,249.7
XS Rating Curve= 0 ,0
Exp/Cntr=0.3,0.1

Type RM Length L Ch R = 1 ,47593.4 ,229.8,231,231.7
XS GIS Cut Line= 2
     2062032.662      181561.105     2062475.371      181222.563
#Sta/Elev= 30
       0 1949.08   104.9  1892.5   121.3 1884.69   137.7 1879.32   150.8 1877.08
   170.5 1875.66   206.5 1874.59   222.9 1875.21   242.6 1874.15   255.7 1874.72
   268.8 1871.33   278.7 1873.04   301.6 1874.02   324.6 1870.91   337.7  1873.8
   350.8 1874.68   367.2 1874.15   382.3 1870.99   396.7 1870.57   406.5 1871.16
   413.1 1872.68   416.4 1874.48   429.5 1886.38   439.3 1892.59   449.1 1896.76
   475.4 1904.82   527.8 1911.57   537.6 1911.06   544.2 1909.46   557.3 1908.63
#Mann= 4 ,-1 , 0
       0     .12       0   382.3    .045       0   406.5     .12       0
   544.2     .06       0
Bank Sta=382.3,406.5
XS Rating Curve= 0 ,0
Exp/Cntr=0.3,0.1

Type RM Length L Ch R = 1 ,47362.4 ,544.3,567.3,588.6
XS GIS Cut Line= 2
     2062197.593      181695.653     2062705.405      181350.601
#Sta/Elev= 30
       0 1890.11    78.4 1876.12  109.49  1874.7   186.1 1875.58   199.2 1874.38
   212.3 1870.94   228.6 1870.18   244.9 1872.28   277.6 1872.53   290.6  1869.7
   316.8 1871.88   342.9 1871.38   353.1  1869.9   362.5 1869.66   375.6 1870.06
   382.1 1871.41   385.4 1873.48   398.4 1885.23   408.2 1895.36   411.5 1897.67
  429.141906.297   440.9 1912.71  452.68 1913.42   489.8 1914.12  500.571913.307
  511.531912.781  536.911911.301   587.8 1907.98   600.9 1904.73     614 1902.94
#Mann= 9 ,-1 , 0
       0     .06       0  109.49     .12       0   353.1    .045       0
   375.6     .12       0  429.14     .06       0  452.68    .016       0
  500.57     .12       0  511.53     .08       0  536.91     .12       0
Bank Sta=353.1,375.6
XS Rating Curve= 0 ,0
Exp/Cntr=0.3,0.1

Type RM Length L Ch R = 1 ,46795.1 ,608,617.8,626.4
XS GIS Cut Line= 3
     2062130.319      181875.775     2062586.048      182051.556
     2062727.107      182023.344
#Sta/Elev= 30
       0  1917.7    42.6 1905.56    78.7 1896.68   95.691891.648   137.7 1877.25
   160.6 1873.44     259 1870.45  331.361871.216   347.5 1871.69   360.6 1871.27
     377 1869.58   390.1 1866.82   396.7 1865.87   416.3 1865.83   426.2 1866.26
   445.8  1869.3   498.3 1881.85   508.1 1884.92   527.7 1892.06   560.4 1905.96
     580  1916.8  588.631923.208   596.3 1929.01   599.6 1930.68   609.4 1931.96
  620.191931.831   622.5 1931.88   625.8 1933.29     629 1936.14   632.3 1940.14
#Mann= 7 ,-1 , 0
       0     .12       0   95.69     .06       0  331.36     .12       0
   390.1    .045       0   416.3     .12       0  588.63    .016       0
  620.19     .12       0
Bank Sta=390.1,416.3
XS Rating Curve= 0 ,0
Exp/Cntr=0.3,0.1

Type RM Length L Ch R = 1 ,46177.3 ,537.7,556.5,574.5
XS GIS Cut Line= 3
     2061926.325      182218.657     2062390.735      182672.216
     2062549.155      182713.449
#Sta/Elev= 30
       0 1921.82     9.8 1917.31      23 1912.36    45.9 1901.02    75.4 1889.56
   101.6 1883.03   132.71878.028   163.9 1871.92   186.9 1868.38   209.8 1866.34
   229.5 1866.35  233.311865.234   239.3 1863.73   265.6 1864.94   287.8 1863.77
   298.4 1862.87   308.2 1863.72  339.461864.743   370.5 1865.82   380.3 1867.07
   514.7 1869.66  675.24 1870.18   708.1 1871.07  714.81 1874.56   721.2  1879.8
   724.4 1881.13   744.1 1881.39  754.231889.152   793.2 1909.36   812.8 1918.24
#Mann= 9 ,-1 , 0
       0     .12       0   132.7     .06       0  233.31     .12       0
   287.8    .045       0   308.2     .12       0  339.46     .06       0
  675.24     .12       0  714.81    .016       0  754.23     .12       0
#XS Ineff= 2 , 0
                           452.8         1876.17
Permanent Ineff=
       F       F
Bank Sta=287.8,308.2
XS Rating Curve= 0 ,0
Exp/Cntr=0.3,0.1

Type RM Length L Ch R = 1 ,45620.9 ,479.1,492.3,502.8
XS GIS Cut Line= 3
     2061618.166      182448.692     2061646.378      182537.667
     2061663.739      183149.646
#Sta/Elev= 30
       0  1925.1     6.4 1923.21    16.1 1922.21    32.2 1916.16    64.4 1900.26
    93.3 1882.89   116.3 1873.36   129.4 1869.94  161.111865.057   181.7 1865.06
   194.8 1862.06   204.6 1860.94   214.5 1861.38  286.48 1862.37   306.2 1862.19
   332.3 1860.58   342.2 1860.83     352 1862.59     388 1863.86     424 1866.27
  457.781869.683   482.9 1873.24  528.511877.818   561.5 1881.26   574.6 1885.58
  621.721886.108   636.8 1887.65   653.2 1890.96   679.4 1893.94   705.6 1901.03
#Mann= 8 ,-1 , 0
       0     .12       0  161.11     .06       0   194.8    .045       0
   214.5     .06       0  286.48     .12       0  457.78     .06       0
  528.51    .016       0  621.72     .06       0
Bank Sta=194.8,214.5
XS Rating Curve= 0 ,0
Exp/Cntr=0.3,0.1

Type RM Length L Ch R = 1 ,45128.5 ,527.7,517.4,506.6
XS GIS Cut Line= 2
     2061331.707      182392.268     2060945.423      183117.094
#Sta/Elev= 30
       0 1933.81    22.9 1924.33    49.1 1911.74    78.5 1896.11    85.1 1891.35
    94.9 1879.64     108 1865.54   111.3 1863.27   121.5 1859.55   130.9 1857.97
     144 1859.25   157.1  1860.6   271.71861.322     301 1860.54   320.7 1861.58
     337 1861.28     373 1864.49   441.8    1864   566.1 1865.25     589 1866.77
   605.4 1870.29  630.861872.726   647.9 1873.82  662.791873.657  670.331875.703
   726.4 1882.78  739.861886.086   752.6 1886.74  775.76 1891.23   821.3 1902.27
#Mann= 9 ,-1 , 0
       0     .12       0   121.5    .045       0     144     .12       0
   271.7     .06       0  630.86    .016       0  662.79     .08       0
  670.33     .06       0  739.86    .016       0  775.76     .06       0
#XS Ineff= 2 , 0
                          431.88         1880.36
Permanent Ineff=
       F       F
Bank Sta=121.5,144
XS Rating Curve= 0 ,0
Exp/Cntr=0.3,0.1

Type RM Length L Ch R = 1 ,44611.1 ,528.1,528.3,525
XS GIS Cut Line= 3
     2060797.853      182166.574     2060789.173      182539.837
     2060602.541        182891.4
#Sta/Elev= 30
       0 1961.71     6.6 1958.38    22.9 1948.72    49.1 1935.79    68.8 1923.97
    91.7 1906.58   101.5 1897.07     131 1872.52   140.8 1866.36   157.2 1857.48
   160.5 1856.68   183.4 1856.34     190 1856.92   196.5 1858.82   203.1 1859.59
   212.9 1858.56   222.7 1858.45   268.6 1867.64   360.11877.879  374.661879.165
  422.991885.288   432.1 1887.43   458.2 1885.89  467.181888.537   474.5 1890.63
   484.3 1892.24  500.621894.022  518.611896.514   683.3 1914.17   771.4    1925
#Mann= 9 ,-1 , 0
       0     .12       0   157.2    .045       0     190     .12       0
   360.1     .06       0  374.66     .12       0  422.99    .016       0
  467.18     .08       0  500.62     .12       0  518.61     .06       0
Bank Sta=157.2,190
XS Rating Curve= 0 ,0
Exp/Cntr=0.3,0.1

Type RM Length L Ch R = 1 ,44082.8 ,898.3,901.2,897.2
XS GIS Cut Line= 4
     2060413.739      182023.344      2060283.53      182212.146
     2060303.062      182637.494     2060376.846      182834.976
#Sta/Elev= 30
       0 1945.26    22.9 1932.31      59 1913.76    85.2  1902.9    98.3 1895.97
     118 1893.25   140.9 1888.67   173.6 1880.45   199.9 1876.77     249 1866.89
   281.8 1861.97   311.2 1859.75   330.9 1859.89   347.3 1855.67   357.1 1855.19
   373.5 1854.29   386.6 1854.62   396.4 1857.04   409.5 1856.18     439 1858.99
  513.621858.049     534 1862.16   551.61862.022   556.9 1862.15   566.7    1864
   596.2 1871.88   684.3 1899.74   771.9 1914.68   807.6 1919.67     866 1926.26
#Mann= 5 ,-1 , 0
       0     .12       0   357.1    .045       0   386.6     .12       0
  513.62    .016       0   551.6     .06       0
#XS Ineff= 2 , 0
                          512.72         1873.14
Permanent Ineff=
       F       F
Bank Sta=357.1,386.6
XS Rating Curve= 0 ,0
Exp/Cntr=0.3,0.1

Type RM Length L Ch R = 1 ,43181.6 ,899.6,883.6,866.1
XS GIS Cut Line= 4
     2059922.745      181753.871     2059819.121      181990.792
     2059836.482      182628.813     2059793.079      182817.615
#Sta/Elev= 30
       0 1891.56      36 1885.24      72 1884.12   134.2 1876.83  174.471874.649
   240.51872.083  294.091868.809     311 1866.95   314.2 1864.92     324 1852.72
   330.6 1851.79   345.1 1852.11  371.991856.321   461.5  1855.9   510.6 1857.86
   651.4  1857.1   703.7 1859.18   762.6 1859.41  777.651862.496   798.7 1862.38
  805.211867.049     815 1874.91   837.9 1886.77   867.4 1904.58   909.8 1923.83
   932.4 1928.43   971.1 1933.55 1025.631932.994  1061.5 1932.62  1090.6 1934.24
#Mann= 10 ,-1 , 0
       0     .12       0  174.47     .08       0   240.5     .06       0
  294.09     .12       0     324    .045       0   345.1     .12       0
  371.99     .06       0  777.65    .016       0  805.21     .12       0
 1025.63     .06       0
#XS Ineff= 2 , 0
                          575.92         1874.05
Permanent Ineff=
       F       F
Bank Sta=324,345.1
XS Rating Curve= 0 ,0
Exp/Cntr=0.3,0.1

Type RM Length L Ch R = 1 ,42298   ,714,717.6,720
XS GIS Cut Line= 3
     2059021.703      182287.725      2059495.77      182785.063
     2059602.107      182845.827
#Sta/Elev= 30
       0  1985.6    45.8 1949.65    58.9 1945.59   111.2 1906.09   150.5 1881.65
   170.1 1870.91   196.3 1861.93   235.6 1854.27   274.8 1853.91  315.531850.006
  321.761850.566     337 1848.72   356.6 1848.22   359.9 1848.35  365.181849.629
   369.7 1851.18  410.581854.903   468.81856.717  539.121855.912  546.851856.053
  664.161856.839  666.121856.852   680.5 1858.53   693.5 1865.69   716.1  1866.8
  722.641869.367   738.6 1881.78   777.3  1900.1  805.651911.096   809.6 1912.16
#Mann= 14 ,-1 , 0
       0     .12       0  315.53     .06       0  321.76     .12       0
     337    .045       0   359.9     .12       0  365.18    .016       0
  410.58     .06       0   468.8     .12       0  539.12     .06       0
  546.85     .12       0  664.16     .06       0  666.12    .016       0
  722.64     .12       0  805.65     .06       0
Bank Sta=337,359.9
XS Rating Curve= 0 ,0
Exp/Cntr=0.3,0.1

Type RM Length L Ch R = 1 ,41580.4 ,439.3,469.4,498.4
XS GIS Cut Line= 2
     2058628.474      182610.642     2059048.721      183264.664
#Sta/Elev= 30
       0 1947.39     9.8 1938.81    26.2 1927.56    42.6 1912.93    55.8 1904.38
    75.4 1888.25    95.1  1867.8   111.5 1847.95   114.8    1845   118.1 1843.68
   127.9 1843.38     141 1844.15   177.1 1849.32     187 1847.98   196.8 1849.12
   209.9 1846.24   219.8  1845.3   226.3 1845.96   242.7 1850.94   249.3 1851.44
  326.161851.076  431.28 1852.25  435.551852.181  470.661852.434  483.121853.125
  507.761854.042   583.9 1854.89   652.8 1858.94  773.991859.199   777.4 1859.35
#Mann= 10 ,-1 , 0
       0     .12       0   118.1    .045       0     141     .12       0
  326.16     .06       0  431.28     .12       0  435.55    .016       0
  470.66     .12       0  483.12    .016       0  507.76     .06       0
  773.99    .016       0
#XS Ineff= 2 , 0
                          263.65         1868.29
Permanent Ineff=
       F       F
Bank Sta=118.1,141
XS Rating Curve= 0 ,0
Exp/Cntr=0.3,0.1

Type RM Length L Ch R = 1 ,41111   ,459.3,461.4,463.2
XS GIS Cut Line= 2
     2058458.444      182637.494     2057996.204      183153.987
#Sta/Elev= 30
       0 1934.17    26.2 1918.37    39.2 1909.13    58.8 1897.85    91.6 1875.04
   104.6 1862.44   107.9 1859.79   124.2 1849.24   130.8 1845.68   147.1 1843.06
   160.2 1844.62   183.1  1845.4   219.1 1843.63   232.1 1844.06   238.7 1843.57
   251.8 1844.27   277.9 1843.21   287.7 1842.37   298.4 1842.79   307.3 1843.81
  316.131847.214   330.2 1852.44   356.4 1857.27   372.7 1861.08   385.8 1862.21
   392.3 1864.14   493.7 1874.18   555.8 1882.93   601.6 1886.14   693.1 1900.73
#Mann= 4 ,-1 , 0
       0     .12       0   277.9    .045       0   298.4    .016       0
  316.13     .12       0
Bank Sta=277.9,298.4
XS Rating Curve= 0 ,0
Exp/Cntr=0.3,0.1

Type RM Length L Ch R = 1 ,40649.6 ,501,532.2,561.8
XS GIS Cut Line= 3
     2058381.078      182376.267     2058141.603      182400.949
     2057766.169      182759.021
#Sta/Elev= 30
       0 1950.92    19.5 1938.84    58.6    1920   143.1 1874.41   175.7 1859.25
   185.4 1856.48   198.4 1854.55   283.2 1848.04   286.4 1846.69     293 1841.05
   296.2 1839.51   309.2 1836.43   315.8 1836.03   328.8  1836.7   341.9 1839.26
   364.7 1838.14   377.8 1839.64   390.8  1839.2   397.4 1841.42  403.031845.125
   420.2 1856.51   426.7 1858.87  437.961860.788   508.3 1869.94   573.6 1881.27
   612.7 1889.22   642.1 1892.97   664.9    1899   713.9 1917.03   759.6 1931.06
#Mann= 5 ,-1 , 0
       0     .12       0   309.2    .045       0   328.8     .12       0
  403.03    .016       0  437.96     .12       0
Bank Sta=309.2,328.8
XS Rating Curve= 0 ,0
Exp/Cntr=0.3,0.1

Type RM Length L Ch R = 1 ,40117.4 ,701.4,699.4,696.2
XS GIS Cut Line= 2
     2058313.044      182207.806     2057740.128      181834.542
#Sta/Elev= 30
       0 1895.27      72  1864.4     108 1857.03  150.621853.531  187.611851.529
   209.4  1848.6   235.6 1841.81   261.7  1842.3   287.9 1839.16   304.3 1831.06
   343.5 1838.41   363.2  1837.9   376.2 1834.81   392.6 1836.04   405.7 1831.02
   431.9 1830.42   438.4 1829.67   451.9 1830.09   461.3 1833.73   464.6 1836.83
   480.9 1864.87   487.5 1872.67   513.7 1890.76   539.8 1903.41   582.4 1918.33
   588.9 1922.43   608.5 1943.88   615.1 1949.06   644.5 1964.57   683.8 1977.62
#Mann= 5 ,-1 , 0
       0     .12       0  150.62    .016       0  187.61     .12       0
   431.9    .045       0   451.9     .12       0
#XS Ineff= 2 , 0
          347.03 1857.14
Permanent Ineff=
       F       F
Bank Sta=431.9,451.9
XS Rating Curve= 0 ,0
Exp/Cntr=0.3,0.1

Type RM Length L Ch R = 1 ,39418   ,520.7,491.7,457.5
XS GIS Cut Line= 3
     2058536.569      181713.015     2058187.176      181526.383
     2057957.141      181582.806
#Sta/Elev= 30
       0 1931.39      36  1923.1    58.9 1913.12    78.6 1913.26    98.2 1903.95
   101.5 1900.55   104.8  1894.9  110.461882.408   114.6 1873.66   117.8  1869.5
   147.61863.113   189.9 1854.38     203 1850.32   209.5 1846.83   216.1 1841.63
   232.4 1823.86   235.7 1821.34   252.1 1817.05   265.2 1816.77   278.3 1816.99
   294.6 1820.68   314.3 1833.65   353.6 1832.33   392.8 1839.27   451.3  1845.6
   480.5 1850.91   506.4 1859.85   535.6 1862.98   555.1 1866.53     633 1885.47
#Mann= 5 ,-1 , 0
       0     .12       0  110.46    .016       0   147.6     .12       0
   252.1    .045       0   278.3     .12       0
Bank Sta=252.1,278.3
XS Rating Curve= 0 ,0
Exp/Cntr=0.3,0.1

Type RM Length L Ch R = 1 ,38926.3 ,468.3,446.7,425.2
XS GIS Cut Line= 3
     2058544.286      181016.056     2058430.232      181038.101
     2058021.972      181428.322
#Sta/Elev= 30
       0 1860.01    22.6 1852.21    74.2 1842.81   96.891839.838   112.9 1836.43
   122.7 1830.09   132.5 1821.55  139.391817.767   158.6 1810.59   165.1 1809.24
   234.7 1806.79   243.5 1806.62   256.5 1807.89   263.1  1812.8   269.6 1815.66
   289.2 1812.59   305.5 1811.47   331.6 1818.29   357.7 1816.27   370.8 1817.82
   383.8 1821.13   419.8 1824.44   426.3 1825.93   442.6 1833.93   458.9 1839.52
   491.6 1844.11   507.9 1843.75     521 1845.63   618.9 1848.76   680.9 1856.84
#Mann= 5 ,-1 , 0
       0     .12       0   96.89    .016       0  139.39     .12       0
   234.7    .045       0   256.5     .12       0
#XS Ineff= 2 , 0
                          269.87         1824.17
Permanent Ineff=
       F       F
Bank Sta=234.7,256.5
XS Rating Curve= 0 ,0
Exp/Cntr=0.3,0.1

Type RM Length L Ch R = 1 ,38479.6 ,528.2,527.7,526
XS GIS Cut Line= 3
     2057894.261      180830.413     2058021.635      181331.138
     2057988.704      181439.947
#Sta/Elev= 30
       0 1950.01    52.3 1910.07    65.4  1902.2    75.2 1895.02   107.9 1878.44
   140.6 1855.48   143.9  1850.5   150.4 1835.35   153.7 1829.88   166.8 1819.11
   186.4 1810.34   202.7 1801.72   215.8 1797.95   225.6 1796.56   284.5 1799.61
   297.6 1799.38   304.1 1798.36   320.5 1798.13     327 1798.84   336.8 1800.92
   346.6 1805.08   353.2 1806.92     399 1808.34   431.6 1810.89   490.5 1824.76
   503.6 1829.22   513.4 1830.95   526.4 1835.31   565.4 1845.74   630.4    1860
#Mann= 3 ,-1 , 0
       0     .12       0   304.1    .045       0     327     .12       0
Bank Sta=304.1,327
XS Rating Curve= 0 ,0
Exp/Cntr=0.3,0.1

Type RM Length L Ch R = 1 ,37951.9 ,764.8,764.2,762.2
XS GIS Cut Line= 2
     2057405.416      181039.443     2057570.112      181569.254
#Sta/Elev= 30
       0 1880.01    42.4  1856.4    65.3 1844.75    75.1 1841.37   137.1 1811.89
   143.6 1806.66   156.7 1793.64   163.2 1789.19   169.7 1788.04     186 1789.46
   202.4 1789.49   215.4 1788.61   240.3 1784.74   251.3  1784.5   264.4 1784.87
   270.9 1787.19   277.4 1791.95   280.7 1792.95   316.6 1791.38   332.9 1792.15
     346 1789.72     359 1790.92   365.5 1792.58   381.8 1802.88   404.7 1815.45
   430.8 1825.73   440.6 1832.85   505.9 1869.79     532 1881.16   554.8 1890.01
#Mann= 3 ,-1 , 0
       0     .12       0   240.3    .045       0   264.4     .12       0
#XS Ineff= 2 , 0
                          287.28         1808.57
Permanent Ineff=
       F       F
Bank Sta=240.3,264.4
XS Rating Curve= 0 ,0
Exp/Cntr=0.3,0.1

Type RM Length L Ch R = 1 ,37187.7 ,729.5,732,732.7
XS GIS Cut Line= 3
     2056748.374      181205.202     2056735.353      181313.709
     2056978.409      181971.261
#Sta/Elev= 30
       0 1852.83    35.4 1829.71    61.1 1814.82    99.6 1797.96   109.3  1790.9
   122.4 1777.69   132.2 1772.98   145.3 1772.83   174.8  1775.9   191.2 1773.46
   233.8 1775.09   250.2 1773.88   266.5 1775.37   298.4 1772.98   312.4 1771.93
  320.19 1773.05   328.8 1775.91   384.5  1776.5   400.8 1773.82   453.2 1772.24
   469.6 1775.36   495.8 1776.89   541.7 1775.87   577.7 1778.11   587.6 1780.75
     617 1796.58   633.4 1802.94   718.6 1822.41   728.4 1822.76   810.3 1847.63
#Mann= 3 ,-1 , 0
       0     .12       0   298.4    .045       0  320.19     .12       0
#XS Ineff= 2 , 0
                          494.63          1795.6
Permanent Ineff=
       F       F
Bank Sta=298.4,320.19
XS Rating Curve= 0 ,0
Exp/Cntr=0.3,0.1

Type RM Length L Ch R = 1 ,36455.6 ,1283.2,1292.5,1294.3
XS GIS Cut Line= 3
     2056201.499      181283.327     2056129.885      181476.469
     2056342.558      182194.785
#Sta/Elev= 30
       0  1804.8     9.8 1800.89    22.9 1800.88   45.161796.779     170 1772.69
   222.4 1766.88   251.8 1761.52   264.9 1760.76   274.7 1757.92   310.7 1760.99
   349.9 1758.43   370.5 1758.41   379.4 1760.55   395.7 1758.62   412.1 1760.13
   448.1 1755.92   474.2 1761.29     556 1756.43   575.6  1757.1   598.6 1760.26
   641.1  1761.5   660.7  1759.2   716.3 1762.66     736 1760.93   758.8 1762.95
   781.8 1760.12   814.5 1761.77   873.4 1776.57   899.5 1781.25   955.1 1798.78
#Mann= 4 ,-1 , 0
       0    .016       0   45.16     .12       0   349.9    .045       0
   370.5     .12       0
#XS Ineff= 2 , 0
                          641.04         1769.93
Permanent Ineff=
       F       F
Bank Sta=349.9,370.5
XS Rating Curve= 0 ,0
Exp/Cntr=0.3,0.1

Type RM Length L Ch R = 1 ,35163.1 ,567.6,581.1,595.3
XS GIS Cut Line= 3
     2055374.676      181350.601     2055123.266      181730.433
     2055201.391      182394.496
#Sta/Elev= 30
       0 1758.51   45.011756.896  107.211755.032  108.251755.005  151.911753.881
  294.881750.431  338.951751.241   488.3 1746.39   504.7 1742.78   517.8 1735.68
   534.2 1732.82   573.5 1734.09   593.2 1733.26   606.3 1734.85   658.7 1736.17
   675.1 1733.11   688.2 1734.18   707.9 1731.75     721 1730.17   724.5 1732.22
   730.8 1733.73   753.8 1730.36   776.7 1734.29   881.6 1739.13   930.8 1744.55
   960.3 1751.58  1012.7 1771.41    1052 1784.49  1084.8 1792.57  1124.1 1798.99
#Mann= 9 ,-1 , 0
       0    .016       0   45.01     .06       0  107.21     .12       0
  108.25     .06       0  151.91     .12       0  294.88    .016       0
  338.95     .12       0   707.9    .045       0   724.5     .12       0
Bank Sta=707.9,724.5
XS Rating Curve= 0 ,0
Exp/Cntr=0.3,0.1

Type RM Length L Ch R = 1 ,34582   ,284.5,276.9,276.8
XS GIS Cut Line= 3
     2055003.582      181276.817     2054591.256       181947.39
     2054586.916      182088.449
#Sta/Elev= 30
       0 1747.04   134.5 1742.66  234.351742.469  292.171742.261   314.9 1741.49
  334.341737.554   383.8 1724.88   419.8 1724.51   436.2  1721.9   449.4 1723.48
     469 1721.24   485.4 1724.76   495.3 1725.02   518.2 1720.53   541.2 1723.55
   606.8 1723.56     633 1719.81   646.2 1719.31   656.5 1720.44   669.1 1723.97
   695.4 1724.01   708.5 1731.88   731.4 1749.57   747.8 1765.24   764.2  1775.9
   803.2 1790.95   841.7 1802.48   851.4 1806.73   899.5 1834.43   928.3 1841.59
#Mann= 6 ,-1 , 0
       0     .06       0  234.35     .12       0  292.17    .016       0
  334.34     .12       0     633    .045       0   656.5     .12       0
Bank Sta=633,656.5
XS Rating Curve= 0 ,0
Exp/Cntr=0.3,0.1

Type RM Length L Ch R = 1 ,34305   ,387.2,395.7,394.8
XS GIS Cut Line= 3
     2054771.812      181159.629     2054359.485      181830.202
     2054355.145      181971.261
#Sta/Elev= 30
       0 1739.58   124.6 1735.92  210.181738.719   236.2 1738.95   285.4 1735.39
   291.9 1734.41     328 1723.77  341.281723.182  356.751721.816   400.2 1722.25
   436.2 1718.81   449.4 1713.99   472.3 1715.88     515  1716.3   528.1 1715.23
   538.5 1717.05   547.8 1718.96   577.3 1719.95   642.9  1717.5   646.2 1718.52
     656 1725.44   662.6 1735.25   669.1 1746.86   672.4 1751.08   701.9 1764.13
     738 1784.03   783.9 1807.34   806.4 1814.53   828.9 1820.03   928.3 1835.77
#Mann= 6 ,-1 , 0
       0     .06       0  210.18     .12       0  341.28    .016       0
  356.75     .12       0     515    .045       0   538.5     .12       0
Bank Sta=515,538.5
XS Rating Curve= 0 ,0
Exp/Cntr=0.3,0.1

Type RM Length L Ch R = 1 ,33909.4 ,319.2,317.5,314.7
XS GIS Cut Line= 3
     2054461.048      180996.869     2054072.593      181630.549
     2054094.294      181895.306
#Sta/Elev= 30
       0 1732.24   128.1 1732.09   160.4 1728.15   173.5 1724.11   189.9 1721.13
  249.41 1718.71     370 1714.28   410.1  1708.9   419.1 1708.04   428.9 1708.58
   435.5 1710.95     478  1710.5   491.2    1713   507.5  1713.7   527.2 1710.61
   586.1 1713.26   651.6 1712.11     668 1713.13   677.8  1717.3   694.2 1729.29
   697.4 1732.41   707.2 1749.75   710.5 1754.34   713.8 1757.03   733.4 1765.96
   753.1 1772.49   785.9 1787.42   831.8 1800.29  935.85 1820.42  1008.9 1827.46
#Mann= 6 ,-1 , 0
       0     .06       0   128.1     .12       0  249.41     .06       0
   410.1    .045       0   428.9     .12       0  935.85     .06       0
Bank Sta=410.1,428.9
XS Rating Curve= 0 ,0
Exp/Cntr=0.3,0.1

Type RM Length L Ch R = 1 ,33591.9 ,333.7,336.9,339.5
XS GIS Cut Line= 3
     2054126.412      180873.605     2053809.572      181535.497
     2053822.593      181724.299
#Sta/Elev= 30
       0 1726.63   111.4  1726.6   137.6 1726.24  147.171725.262  214.831718.463
  226.391718.219   330.9 1715.52     380 1718.54   383.3  1717.7   386.6 1714.58
   393.1 1705.93   396.4 1704.24   406.2 1703.85   423.4 1704.98     439 1703.97
   445.5 1704.96   455.4 1707.37   471.7 1708.98   550.4 1707.16   615.9  1709.4
  646.431709.011  651.061709.195   671.6 1709.66   681.4 1711.31   714.2 1723.54
   756.7 1742.09   799.1 1763.98   851.3 1786.75   874.1 1792.26   923.1  1799.8
#Mann= 8 ,-1 , 0
       0     .06       0  147.17     .12       0  214.83     .06       0
  226.39     .12       0   423.4    .045       0   445.5     .12       0
  646.43     .06       0  651.06     .12       0
Bank Sta=423.4,445.5
XS Rating Curve= 0 ,0
Exp/Cntr=0.3,0.1

Type RM Length L Ch R = 1 ,33255   ,630.3,642.9,653.9
XS GIS Cut Line= 3
     2053848.536      180791.704     2053454.018      181410.449
     2053444.123       181599.44
#Sta/Elev= 30
       0 1722.39   196.6 1723.47  231.311722.828   242.4 1722.03     249 1720.67
   252.2 1719.17   265.4 1707.36   275.2 1700.77   278.5 1699.34   281.7 1698.74
   298.1 1698.29   310.9 1699.16   334.2 1703.71   350.5 1703.91   373.5 1701.94
   393.1 1701.24  407.971701.891   442.3 1703.84   589.7 1704.73   655.2 1705.95
  667.741706.723  691.991709.133   714.2 1712.32   737.1 1718.74  745.811722.838
   779.5 1736.36   805.6 1744.94   831.7 1751.68   857.8 1755.74   923.1 1761.01
#Mann= 8 ,-1 , 0
       0     .06       0  231.31     .12       0   278.5    .045       0
   310.9     .12       0  407.97     .06       0  667.74     .08       0
  691.99     .06       0  745.81     .12       0
#XS Ineff= 2 , 0
                          416.05         1713.33
Permanent Ineff=
       F       F
Bank Sta=278.5,310.9
XS Rating Curve= 0 ,0
Exp/Cntr=0.3,0.1
